HEC-RAS study LTTLRV1.prj: LTTLRV1

--- LTTLRV1.g01 (geometry) --- (continued)

Type RM Length L Ch R = 1 ,34557   ,289.9,284.5,280.4
XS GIS Cut Line= 2
2329962.15194798603694.2680585252330027.00702808604110.005751474
#Sta/Elev= 30
       0 3229.61    15.1 3226.06    47.5 3216.69    55.6 3213.51    63.7 3208.18
    67.7 3207.01    79.9 3206.97   100.1  3199.5   119.9 3197.76   128.4 3195.88
   160.8    3195     173 3196.27   189.2 3194.81   217.5 3195.74   229.7 3197.02
   245.8 3195.62     262 3197.05   290.4 3195.66   314.7 3195.64   333.5 3192.38
     351 3190.88   363.3 3191.37   367.3 3192.55   371.3 3194.88   379.4 3201.71
   391.6 3215.41   400.1 3219.29   407.8 3224.59   411.8 3225.62   420.8 3225.91
#Mann= 5 ,-1,0
       0      .1       0      60     .06       0     160      .1       0
   333.5    .045       0   367.3     .06       0
#XS Ineff= 2 , 0
           175.7 3204.07
Permanent Ineff=
       F       F
Bank Sta=333.5,367.3
XS Rating Curve= 0 ,0
Exp/Cntr(USF)=0,0
Exp/Cntr=0.3,0.1

Type RM Length L Ch R = 1 ,34272   ,198.4,189.8,183.8
XS GIS Cut Line= 2
2329612.40878765603731.1206370462329772.87315061604199.750747184
#Sta/Elev= 30
       0 3222.17    14.9 3216.64    23.3 3212.41    58.1 3200.56    95.2 3192.73
   112.1 3192.02   196.8 3193.47   230.5 3189.67   243.2  3189.3   281.2 3192.58
   306.6 3191.19   319.5 3192.28   336.2 3191.59   353.1  3192.6   357.3 3191.94
   363.6 3188.02   365.8  3186.7   373.1 3186.32   391.2 3186.44   398.3 3188.06
   403.8 3189.63     425 3189.96   433.4 3191.08   442.4 3196.79   454.6 3206.67
     463  3211.1   471.5 3214.11   479.9 3219.61   484.2 3220.96   495.3 3221.77
#Mann= 7 ,-1,0
       0      .1       0     130     .06       0     240     .12       0
     340      .1       0   363.6    .045       0   398.3      .1       0
  495.34     .06       0
Bank Sta=363.6,398.3
XS Rating Curve= 0 ,0
Exp/Cntr=0.3,0.1

Type RM Length L Ch R = 1 ,34082   ,159.8,163.2,164.8
XS GIS Cut Line= 3
2329328.79620404603928.7640574412329476.78226136604043.343412059
2329630.95662039604268.135000244
#Sta/Elev= 30
       0 3221.42    33.3 3207.67    45.5  3204.5      66 3193.86    80.2 3191.13
    90.3 3187.85    99.6 3185.94   133.9    3185   151.1 3187.29   193.2 3188.08
   208.8 3184.64   218.5 3184.12   237.9 3186.09   254.2 3187.06   262.8  3186.8
     278 3188.65   296.1 3186.77   305.8 3186.85   314.6 3185.95   339.7  3185.5
   348.7 3186.02   363.5 3186.28   378.5 3184.88   405.3 3186.13   412.5 3189.38
   421.1 3196.06   432.6 3202.41   446.5 3207.47   456.2 3209.34   459.7 3210.97
#Mann= 7 ,-1,0
       0      .1       0      40     .06       0  197.16     .12       0
   314.6    .045       0   348.7     .12       0  367.16      .1       0
  437.16     .06       0
#XS Ineff= 2 , 0
          161.65 3194.81
Permanent Ineff=
       F       F
Bank Sta=314.6,348.7
XS Rating Curve= 0 ,0
Exp/Cntr(USF)=0,0
Exp/Cntr=0.3,0.1

Type RM Length L Ch R = 1 ,33919   ,206.4,195.4,186.6
XS GIS Cut Line= 3
2329245.29194956604054.9673764982329340.77871429604097.510984546
2329510.00773297604408.552030059
#Sta/Elev= 30
       0 3231.45     7.5 3227.79    16.3 3222.17    25.1 3220.06    42.6 3209.02
    55.7 3204.03    60.1 3201.79    68.8 3195.63    76.6 3192.01   113.3 3182.65
     120 3182.31   140.6 3184.43   154.2 3181.78   167.9  3183.3     177 3182.36
   190.7 3183.56   213.4 3182.51   232.13183.713   272.13183.456   286.7  3184.1
   313.6 3182.52   331.8 3182.19   345.7 3183.12   378.1 3181.98   381.9 3183.33
     391 3190.21   413.8 3195.73     443 3205.05   451.8 3208.72   458.6 3209.66
#Mann= 6 ,-1,0
       0      .1       0      40     .06       0  184.54     .12       0
   232.1    .045       0   272.1     .12       0  394.54     .06       0
Bank Sta=232.1,272.1
XS Rating Curve= 0 ,0
Exp/Cntr(USF)=0,0
Exp/Cntr=0.3,0.1

Type RM Length L Ch R = 1 ,33724   ,115.6,114.7,114.1
XS GIS Cut Line= 2
2329146.40454252604252.5214543952329468.54544297604461.446168819
#Sta/Elev= 30
       0 3216.53    10.4 3211.71    16.4 3210.04    25.9 3205.25    39.4  3199.9
    67.4 3190.16    74.1 3188.36    82.7 3183.87    91.4 3181.77    98.7 3178.16
   102.2 3176.94   111.7    3176   116.5 3176.25   121.3 3178.29   126.1 3180.28
   133.5 3181.04   146.4 3180.51   159.4 3178.95   183.3 3181.12   235.7 3182.15
   264.3 3181.64   273.6 3181.27   283.4 3179.99   293.8 3179.97     312 3184.77
   351.7 3197.82   360.4 3201.16   371.9 3207.18   376.1 3208.03     384 3208.21
#Mann= 6 ,-1,0
       0     .06       0      50      .1       0    98.7    .045       0
   121.3      .1       0     160     .12       0     280     .06       0
Bank Sta=98.7,121.3
XS Rating Curve= 0 ,0
Exp/Cntr(USF)=0,0
Exp/Cntr=0.3,0.1

Type RM Length L Ch R = 1 ,33609   ,179.2,201.9,222.1
XS GIS Cut Line= 2
2329131.81373294604381.7322822262329400.96300647604541.920676354
#Sta/Elev= 30
       0 3191.44    23.7 3186.58    28.3 3184.05      33 3180.81    42.3 3176.23
      47  3174.5    51.6 3174.07    64.1 3174.35    72.8 3175.82    79.6 3176.67
     102 3176.38   107.5 3176.96   116.2 3177.02   126.1 3177.97   148.7 3176.93
   160.4 3177.55   178.8 3179.44   186.6 3179.84   192.5 3179.81     210 3178.16
   225.7 3179.41   230.4 3180.53   239.1 3184.68   259.6 3188.78   284.4 3196.58
   291.7 3199.39   298.3 3203.12   300.4 3203.85   303.9 3204.56   313.2 3204.69
#Mann= 5 ,-1,0
       0     .06       0    42.3    .045       0    72.8     .12       0
     120      .1       0     180     .06       0
Bank Sta=42.3,72.8
XS Rating Curve= 0 ,0
Exp/Cntr(USF)=0,0
Exp/Cntr=0.3,0.1

Type RM Length L Ch R = 1 ,33407   ,268.7,291.2,306.9
XS GIS Cut Line= 3
2329058.83788069604425.8385901152329051.44739917604486.515899198
2329110.60907958604781.265692846
#Sta/Elev= 30
       0 3188.86    11.4 3187.78    43.7 3183.41    76.1 3183.28    80.2 3182.62
      84 3181.32    92.4 3177.63   100.6 3174.71   104.6  3173.9   112.8 3174.05
     121 3173.08   129.1 3171.66   137.3  3171.5   145.3 3171.71   152.3 3172.85
   169.9 3174.11   182.2 3172.34   189.7 3173.74   210.7 3175.81     227 3173.35
   239.3 3173.37   254.3 3174.29   259.7 3173.76   284.2 3178.72   315.4 3181.73
   324.9 3181.12   333.1 3181.39   337.2 3182.14   349.4 3185.72   361.8  3186.6
#Mann= 5 ,-1,0
       0     .06       0      20      .1       0     121    .045       0
   152.3      .1       0  321.13     .06       0
Bank Sta=121,152.3
XS Rating Curve= 0 ,0
Exp/Cntr=0.3,0.1

Type RM Length L Ch R = 1 ,33116   ,324.1,313.9,303.9
XS GIS Cut Line= 3
2328904.79236761604383.0836255652328820.60922942604514.442722186
2328691.29259548604676.847338806
#Sta/Elev= 30
       0 3195.09    21.5 3188.44    30.9 3184.18    36.7 3179.84    45.2 3170.62
      50 3167.03    54.7 3165.59    59.5  3165.3      69 3165.52    80.33166.992
   116.5 3169.42   130.8 3168.53   149.8 3170.06   154.5 3169.67   164.6 3166.57
   174.9  3167.4   183.9 3169.02   210.6 3168.54   220.9 3166.78   231.1 3167.68
   241.3 3170.01     253 3170.56   261.8  3169.1     272 3169.65   282.2 3165.92
   287.3 3164.73   303.5 3166.04   317.7 3173.41   333.4 3176.91   363.6 3179.56
#Mann= 5 ,-1,0
       0     .06       0      40      .1       0      50    .045       0
    80.3      .1       0  316.02     .06       0
Bank Sta=50,80.3
XS Rating Curve= 0 ,0
Exp/Cntr(USF)=0,0
Exp/Cntr=0.3,0.1

Type RM Length L Ch R = 1 ,32802   ,230.8,226.2,222.1
XS GIS Cut Line= 3
2328578.49093486604284.1057902232328534.37695284604565.268619759
 2328536.9221882604636.827011784
#Sta/Elev= 30
       0 3196.38     9.2 3193.66      24 3187.09    29.4 3184.26    37.5 3180.56
    41.6 3178.38    49.7 3172.32    61.8 3164.69    65.9 3162.73    69.9 3161.73
    90.2 3160.65    97.5 3159.31   102.3 3158.79   114.5 3158.53   122.6 3158.86
   123.4 3159.15   138.8 3164.32   150.9 3166.18     163 3166.32   171.1 3165.51
   195.4 3163.91   207.6 3164.14   227.8 3165.83     248 3165.97   258.5 3166.98
   279.5 3168.02   320.5 3173.24   332.4 3174.28   340.7 3176.07   356.2 3177.71
#Mann= 4 ,-1,0
       0     .06       0      70      .1       0    97.5    .045       0
   123.4      .1       0
Bank Sta=97.5,123.4
XS Rating Curve= 0 ,0
Exp/Cntr=0.3,0.1

Type RM Length L Ch R = 1 ,32576   ,292.1,298.3,302.2
XS GIS Cut Line= 4
2328364.74150229604225.7896688792328336.96524586604283.840713724
2328348.17154367604535.2639502592328401.63358174604642.188026393
#Sta/Elev= 30
       0 3192.81    10.6  3189.6    25.9 3183.22    34.8 3178.67    48.1  3174.3
    69.7 3162.33    77.7 3160.03    85.7 3156.87    93.7 3155.69    97.7 3157.19
   101.7 3157.44   121.7 3156.57   133.8 3155.84   145.8  3156.4   169.8 3156.42
   181.8 3158.12   197.8 3161.59   201.8  3161.9   217.8 3161.03   233.9 3161.54
   241.9 3159.73   249.9 3159.61   261.9 3162.39   281.9 3162.99     345 3169.02
   368.1 3172.83   385.3 3174.32   416.6 3179.72   425.5 3182.05   435.6 3182.65
#Mann= 6 ,-1,0
       0     .06       0   121.7    .045       0   145.8      .1       0
  326.03     .06       0  426.03      .1       0  435.57     .06       0
#XS Ineff= 2 , 0
                          201.81         3166.46
Permanent Ineff=
       F       F
Bank Sta=121.7,145.8
XS Rating Curve= 0 ,0
Exp/Cntr(USF)=0,0
Exp/Cntr=0.3,0.1

Type RM Length L Ch R = 1 ,32278   ,356.5,353.2,348.4
XS GIS Cut Line= 2
2328082.91671244604167.208371199 2328004.0779368604502.895354192
#Sta/Elev= 30
       0 3186.17    22.6 3177.65      39 3168.27    51.3 3162.81    60.5 3156.03
    67.8 3154.53    77.1 3153.78    84.9 3152.01    88.3 3150.59    92.4 3150.17
   123.7 3150.53   130.93151.451   141.7 3152.31   149.9 3152.16   154.1 3153.02
   158.2  3155.2   162.3 3156.21   174.6 3156.78     191 3156.42   211.6 3154.25
   223.9 3155.06   236.2 3154.57   246.8 3154.97     265 3154.11   273.2 3152.55
   289.6 3152.43     302 3156.49   318.4 3163.36   326.6 3167.71   344.8 3168.55
#Mann= 4 ,-1,0
       0     .06       0    84.9    .045       0   130.9      .1       0
     290     .06       0
#XS Ineff= 2 , 0
                          193.62         3163.07
Permanent Ineff=
       F       F
Bank Sta=84.9,130.9
XS Rating Curve= 0 ,0
Exp/Cntr=0.3,0.1

Type RM Length L Ch R = 1 ,31925   ,103.7,84.1,69.3
XS GIS Cut Line= 2
2327727.00037933604072.1925807732327692.33521722 604398.88547221
#Sta/Elev= 30
       0 3178.99       9 3174.37    13.1 3171.14    21.1 3163.84    32.6 3152.16
    37.2 3148.36    41.2  3146.2    50.7 3144.93    53.3 3144.93    65.4 3147.34
   105.6 3148.76   117.6 3150.51   137.8 3149.65  144.96 3146.63   149.8 3145.54
   165.9 3145.58   169.9 3145.74   174.33146.843     186 3147.82   206.1 3146.08
   230.3 3148.37   250.4 3148.72   262.5  3146.4   268.9  3147.2   278.5 3149.83
   282.6 3150.29   301.7 3151.14   314.7 3150.73   318.8 3152.42   328.5 3157.92
#Mann= 6 ,-1,0
       0      .1       0      80     .06       0  144.96    .045       0
   174.3     .06       0     180      .1       0     210     .06       0
Bank Sta=144.96,174.3
XS Rating Curve= 0 ,0
Exp/Cntr(USF)=0,0
Exp/Cntr=0.5,0.3

Type RM Length L Ch R = 1 ,31840   ,41.7,43.3,42.9
XS GIS Cut Line= 4
2327541.25349007604028.822595139 2327528.1488656604100.501489298
2327674.38075368604307.7264103022327674.83609023604397.512811893
#Sta/Elev= 30
       0 3171.16    16.6 3160.82    32.9 3153.53    49.2 3143.89    53.2  3142.2
    57.3 3141.56    63.1 3142.72    73.7 3146.48    88.4 3147.58   132.4 3147.78
   197.8 3146.15   215.7 3146.64   220.6  3146.3   225.3 3144.93   230.4 3143.93
   240.1 3143.91   248.5 3144.08   253.3 3145.06   264.6  3147.4     281 3147.57
   308.7 3146.26   314.5 3146.89   318.5 3148.39   323.4 3148.75   339.9 3148.16
   371.9 3149.69   387.9 3149.39   391.9 3150.48   403.9 3156.86   416.3 3160.35
#Mann= 5 ,-1,0
       0      .1       0      20     .06       0  132.87     .07       0
   225.3    .045       0   253.3     .06       0
#XS Ineff= 3 ,-1
      36     105    3150     105     214    3146     262     370  3145.6
Permanent Ineff=
       F       F       F
Bank Sta=225.3,253.3
XS Rating Curve= 0 ,0
Exp/Cntr(USF)=0,0
Exp/Cntr=0.5,0.3

Type RM Length L Ch R = 1 ,31797   ,125,140.9,159.5
XS GIS Cut Line= 5
2327513.29393522604015.6411114132327489.35554999604132.021058226
 2327559.0919901604210.9469074272327631.19361017604324.775345135
2327640.89193907604396.300520781
#Sta/Elev= 30
       0 3169.68    13.8    3163    30.2 3154.03    46.5 3146.87    49.7 3146.41
    62.8 3146.15    73.4 3147.96    91.4 3148.24   103.7 3147.15   115.9 3143.27
     131 3142.63   141.2 3143.12     150 3143.46   211.1  3144.7   238.1 3146.52
   243.9  3146.1   249.7 3144.13   258.4 3143.56   296.1 3144.07   301.9 3144.35
   313.5  3146.3   325.1 3146.75   363.3  3147.3   371.4 3145.46   375.4 3145.39
     385 3146.89   391.6 3149.02   407.7 3156.48   423.6 3167.61   431.1 3171.33
#Mann= 7 ,-1,0
       0      .1       0    30.2     .06       0   141.2      .1       0
     150     .07       0   249.7    .045       0   296.1      .1       0
   325.1     .06       0
#XS Ineff= 4 ,-1
      38      87    3152  103.83     245  3145.6  298.58  339.58  3145.2
     348     400    3152
Permanent Ineff=
       F       F       F       F
Bank Sta=249.7,296.1
XS Rating Curve= 0 ,0
Exp/Cntr(USF)=0,0
Exp/Cntr=0.5,0.3

Type RM Length L Ch R = 1 ,31656   ,193.7,207.6,219.7
XS GIS Cut Line= 3
2327507.43548087604017.7024903752327448.62862296  604194.0458779
2327443.34621137604343.478478869
#Sta/Elev= 30
       0 3167.49     8.5 3163.28    20.5 3156.79      29 3152.71    41.6 3145.43
    45.8 3144.35    62.7 3147.62    79.6 3148.04    92.2 3146.97   103.3 3143.53
   109.1 3142.87   122.3 3142.94   142.8 3142.33   150.8 3142.91     162 3144.37
   176.5 3145.21     209 3145.67   233.1 3144.49   241.1 3141.65   245.1 3141.02
   249.1 3140.97   269.1  3141.5   282.1 3142.37   285.1 3143.37   289.1 3145.44
   297.1 3147.64   305.1 3151.99   313.1 3154.15   329.1 3161.52   335.4 3163.49
#Mann= 4 ,-1,0
       0     .06       0     140      .1       0   241.1    .045       0
   269.1      .1       0
#XS Ineff= 2 , 0
           69.66 3159.38
Permanent Ineff=
       F       F
Bank Sta=241.1,269.1
XS Rating Curve= 0 ,0
Exp/Cntr=0.3,0.1

Type RM Length L Ch R = 1 ,31449   ,193.2,198.5,195.9
XS GIS Cut Line= 2
2327418.84809733603956.9466736362327201.87569628604280.278094807
#Sta/Elev= 30
       0 3170.23    19.2 3159.64    36.7 3145.95    40.7 3144.08    48.5 3142.06
    53.3 3141.84    62.6 3144.23    77.4 3144.45      87  3143.7    97.2 3139.99
   108.8 3138.22   120.3 3140.28   135.2 3140.74   173.7  3137.6   177.9 3138.04
   188.1 3141.63     193 3141.93   212.2 3138.62   221.2 3139.62   273.1 3140.77
   287.5 3138.62   308.6 3138.35   313.2 3139.27   316.3 3141.69     323 3148.83
   330.7 3153.55   365.3  3166.2   371.2 3169.53   382.6 3174.19   389.4 3175.95
#Mann= 4 ,-1,0
       0     .06       0     120      .1       0   287.5    .045       0
   313.2      .1       0
#XS Ineff= 2 , 0
           72.66 3160.79
Permanent Ineff=
       F       F
Bank Sta=287.5,313.2
XS Rating Curve= 0 ,0
Exp/Cntr(USF)=0,0
Exp/Cntr=0.3,0.1

Type RM Length L Ch R = 1 ,31250   ,330,325.5,321.8
XS GIS Cut Line= 2
2327360.46962804603866.4550454312327080.15609086604164.446169838
#Sta/Elev= 30
       0 3190.76    14.7  3180.6    25.7 3175.49    44.6 3163.38    58.7 3155.86
    72.9 3144.37    81.4 3138.89    86.1 3137.05    97.1 3137.38   105.5 3139.68
   112.5 3140.53   132.3 3140.17   146.5  3140.6   158.1 3141.87   174.8 3141.81
   193.1 3140.68   201.4 3139.15   212.4 3135.83   216.4 3134.76   223.4 3134.51
   239.8 3134.59   245.6 3135.47   256.8 3136.88   274.8 3137.23   310.6 3135.75
   322.3 3138.63   344.9 3140.49   356.5 3144.24   388.2 3149.63   409.1 3150.82
#Mann= 3 ,-1,0
       0     .06       0   212.4    .045       0   245.6      .1       0
#XS Ineff= 2 , 0
          121.26 3161.09
Permanent Ineff=
       F       F
Bank Sta=212.4,245.6
XS Rating Curve= 0 ,0
Exp/Cntr=0.3,0.1

Type RM Length L Ch R = 1 ,30925   ,125.6,125.7,126.5
XS GIS Cut Line= 2
2327085.12381344603648.5563691962326832.18900105604012.243702986
#Sta/Elev= 30
       0 3172.35     9.8 3167.39    21.2 3160.08    32.7 3155.43    47.1 3148.25
    73.8 3131.74    78.7 3130.31   116.1 3130.44   132.3 3132.41   141.8 3132.81
   176.8 3131.86   190.8    3133   199.4 3131.91   219.5 3132.34   229.8 3131.36
   254.1 3132.68   265.5 3130.55   285.6 3129.49     298 3129.12   316.9 3129.66
     323  3133.2   325.9 3134.03   344.9  3135.9     359  3136.5   366.2  3137.7
   397.7  3146.9   406.3 3148.82     429 3151.22   435.1 3152.68     443 3152.68
#Mann= 6 ,-1,0
       0      .1       0      10     .06       0     120     .07       0
     130      .1       0   285.6    .045       0   316.9      .1       0
#XS Ineff= 2 , 0
          141.55  3146.8
Permanent Ineff=
       F       F
Bank Sta=285.6,316.9
XS Rating Curve= 0 ,0
Exp/Cntr(USF)=0,0
Exp/Cntr=0.3,0.1

Type RM Length L Ch R = 1 ,30799   ,235.2,239.3,242.9
XS GIS Cut Line= 2
2326997.66637764603555.3350136552326740.70298503 603925.46440368
#Sta/Elev= 30
       0 3163.69    16.6  3155.8    23.7 3153.21    51.7 3139.65    68.5 3134.44
    85.7  3130.6   104.5 3130.56   119.1 3128.36   128.9 3128.38   140.4  3130.7
   153.2 3130.88   162.9 3130.33   169.1 3128.24     178 3128.53     192 3127.38
   201.9  3127.3   211.6 3129.03   227.1 3129.97     236  3129.3   240.9 3127.51
   270.1 3129.72   297.2 3127.58   318.2 3127.22   323.6 3127.56   333.4 3129.14
   343.1 3134.94   352.8 3136.27   362.6  3139.9   402.4 3143.49   450.6 3146.41
#Mann= 5 ,-1,0
       0      .1       0     130     .07       0     140      .1       0
   297.2    .045       0   323.6      .1       0
#XS Ineff= 2 , 0
          145.41 3138.68
Permanent Ineff=
       F       F
Bank Sta=297.2,323.6
XS Rating Curve= 0 ,0
Exp/Cntr(USF)=0,0
Exp/Cntr=0.3,0.1

Type RM Length L Ch R = 1 ,30560   ,146.5,149.2,151.2
XS GIS Cut Line= 2
 2326874.2899143603422.5989565422326596.05471766603802.938812499
#Sta/Elev= 30
       0 3150.81      23 3140.82    30.7 3139.24    46.3 3133.38    57.7 3131.13
    80.6 3128.77   107.3 3127.18   117.2 3125.72   132.2 3126.01   140.7  3127.4
   171.7 3128.17   181.6 3127.41   203.7 3127.36   206.4 3127.06   212.3  3124.6
     218 3123.56   227.2  3124.3   274.6 3124.92   300.6  3124.6   315.2 3126.75
   340.2 3125.65   349.7 3127.66   355.1  3127.3   361.1 3125.47   372.6 3125.22
   381.2    3127   389.7 3131.21   399.7 3134.63   429.8 3140.84   471.2 3148.27
#Mann= 5 ,-1,0
       0      .1       0     100     .06       0   212.3    .045       0
   227.2     .06       0     260      .1       0
#XS Ineff= 2 , 0
          167.63 3134.64
Permanent Ineff=
       F       F
Bank Sta=212.3,227.2
XS Rating Curve= 0 ,0
Exp/Cntr(USF)=0,0
Exp/Cntr=0.3,0.1

Type RM Length L Ch R = 1 ,30410   ,259.2,262.1,263.8
XS GIS Cut Line= 2
2326811.82735549 603307.293676772326459.32247927603693.914839362
#Sta/Elev= 30
       0 3155.78    29.6 3143.53    54.9 3134.31    94.6 3127.62     103 3125.75
   114.3  3124.2   130.1 3123.71   156.8  3125.2   170.4 3125.11   195.4  3123.1
   208.2 3125.75   241.8 3124.82   258.7  3124.9   270.1 3122.67   278.6 3121.02
     284 3120.54   289.4 3121.35   292.7 3122.48   296.3 3123.59   301.2 3124.08
   327.3 3123.18     341 3121.72   359.8 3121.35   380.5 3124.41   409.1 3121.29
     421 3121.44   430.2 3124.06   444.8 3130.26   462.7 3134.83   523.2 3155.86
#Mann= 5 ,-1,0
       0      .1       0      80     .06       0     210      .1       0
   270.1    .045       0   292.7      .1       0
#XS Ineff= 2 , 0
          211.01  3133.3
Permanent Ineff=
       F       F
Bank Sta=270.1,292.7
XS Rating Curve= 0 ,0
Exp/Cntr=0.3,0.1

Type RM Length L Ch R = 1 ,30148   ,355.2,374.2,384.3
XS GIS Cut Line= 2
 2326660.2706787603138.7054572652326300.62431528603461.983087301
#Sta/Elev= 30
       0 3146.38     7.5 3144.17    18.8 3138.76    30.1 3135.75    48.5 3127.79
    57.6 3125.73    69.5 3121.93    91.6 3117.95   120.8 3120.85   147.3 3120.26
   193.8 3121.41   219.1 3119.56   231.1 3120.23   279.8 3121.09   285.1  3120.2
   287.5 3118.86   290.9 3117.49   301.3 3117.33   306.7 3117.61   313.4 3118.79
   324.7 3119.18     339 3117.56   361.5  3118.4   419.6 3117.68   423.9  3119.1
   430.4 3123.42   451.9 3133.93   464.4 3137.09   473.4 3140.04   483.6 3144.87
#Mann= 5 ,-1,0
       0      .1       0      40     .06       0     190      .1       0
   287.5    .045       0   313.4      .1       0
#XS Ineff= 2 , 0
          139.13 3134.79
Permanent Ineff=
       F       F
Bank Sta=287.5,313.4
XS Rating Curve= 0 ,0
Exp/Cntr(USF)=0,0
Exp/Cntr=0.3,0.1

Type RM Length L Ch R = 1 ,29774   ,246,249.5,252.1
XS GIS Cut Line= 3
2326540.81924248603012.0412874422326463.15323639603065.892883309
2326124.53436663603165.499890034
#Sta/Elev= 30
       0 3133.63    15.7 3129.16    25.1 3124.92    35.8 3121.69    51.1  3118.5
      76 3115.74    84.6 3117.53    93.3 3117.81   101.8 3117.27   110.1 3114.81
   122.6 3113.61   168.5 3115.68     181 3115.25   189.8 3113.41   214.4 3112.78
   226.9 3112.99   239.4 3115.26   251.9 3115.95   301.9 3116.46   331.1 3114.79
   347.6 3116.46   368.6  3115.3   375.73113.762   393.6 3112.49   406.2  3112.6
   412.93114.108   418.7 3117.38   424.9 3122.49   443.7 3142.15   447.5 3144.41
#Mann= 5 ,-1,0
       0      .1       0   94.51     .06       0  244.51      .1       0
   375.7    .045       0   412.9      .1       0
#XS Ineff= 2 , 0
           92.75 3128.18
Permanent Ineff=
       F       F
Bank Sta=375.7,412.9
XS Rating Curve= 0 ,0
Exp/Cntr=0.3,0.1

Type RM Length L Ch R = 1 ,29525   ,249.3,235,221.3
XS GIS Cut Line= 4
 2326418.7265063 602826.09205337  2326369.946617602863.416059581
 2326130.4573115 602908.079712422325994.25971836603053.795266502
#Sta/Elev= 30
       0  3133.3    48.5 3119.12    57.7 3117.43    67.9 3115.79     108 3115.76
   120.2 3114.14   128.3 3111.97     133 3109.69   140.5 3108.98   193.4 3112.14
   217.8 3111.94   234.1 3110.51   250.4 3110.58   254.5 3109.72   274.8 3109.01
   289.2 3109.85   299.2 3112.31   308.4 3113.03   335.7 3112.66   349.4 3110.66
   366.8 3112.35   378.7 3109.82   405.1 3109.59   426.3 3110.42   437.9 3114.75
     449 3116.35   459.9 3119.92   465.9  3120.3   487.2 3130.46   504.5 3136.03
#Mann= 4 ,-1,0
       0     .06       0  111.42      .1       0   254.5    .045       0
   289.2      .1       0
Bank Sta=254.5,289.2
XS Rating Curve= 0 ,0
Exp/Cntr(USF)=0,0
Exp/Cntr=0.3,0.1

Type RM Length L Ch R = 1 ,29290   ,284.9,276.6,268.5
XS GIS Cut Line= 2
 2326211.4556796 602619.115729662325809.09567084602923.524492282
#Sta/Elev= 30
       0 3122.38     4.1 3121.85    19.2 3122.41    32.4 3121.26    44.2 3113.64
    59.3 3109.66    64.3  3107.1    72.3 3105.64    94.4 3105.74   104.4 3106.81
   123.7 3107.59     138 3106.84   149.6 3109.37   169.2 3109.48   189.1 3108.52
   204.7 3110.19   228.8 3110.64     300 3109.58   321.6 3107.75   335.2 3108.55
   365.3 3108.52     375 3107.04   387.9 3107.48   409.3 3105.54   423.6 3108.57
   440.5 3115.38   460.6 3120.82   470.6 3125.72   480.8 3128.86   504.5 3138.49
#Mann= 3 ,-1,0
       0     .06       0    64.3    .045       0   104.4      .1       0
Bank Sta=64.3,104.4
XS Rating Curve= 0 ,0
Exp/Cntr=0.3,0.1

Type RM Length L Ch R = 1 ,29013   ,288.5,288.1,287.2
XS GIS Cut Line= 2
2326009.31339964602405.3325583132325691.09442479602832.361892303
#Sta/Elev= 30
       0 3142.11    26.4  3141.1    54.7 3134.48    63.6 3131.56    72.2 3126.58
    89.6  3111.9      95 3109.54   106.5 3106.92     115 3102.06   119.5 3101.02
   134.5 3100.91   146.5 3101.81   154.5 3103.79   166.5 3105.18   180.8 3105.62
   235.1 3101.48   249.6  3105.4   263.7 3106.14   314.1 3106.17   336.6  3102.6
   349.4 3102.65     358 3104.23   376.8 3105.08   386.6 3103.55   403.9 3102.58
   426.6 3105.72   453.8 3107.89   477.2 3112.01   508.6 3122.38   532.6 3133.39
#Mann= 3 ,-1,0
       0     .06       0     115    .045       0   146.5      .1       0
Bank Sta=115,146.5
XS Rating Curve= 0 ,0
Exp/Cntr(USF)=0,0
Exp/Cntr=0.3,0.1

Type RM Length L Ch R = 1 ,28725   ,230.2,233.5,237.3
XS GIS Cut Line= 2
2325782.62169979602224.9238047522325477.10268229602649.772533242
#Sta/Elev= 30
       0    3130    10.5 3129.48    15.1 3128.35    24.9 3121.44    34.8 3116.61
    52.1 3105.63      59 3102.86      89  3100.2   108.7  3102.3   123.5 3099.93
   134.4 3100.08   148.1 3098.47   148.1 3098.46   154.9 3097.46   172.8 3098.13
   191.1 3097.65   222.6 3099.62   256.5  3098.6   266.4 3099.81   288.6  3100.2
   305.7 3098.59   315.6 3099.02   325.5 3096.82   334.4 3097.19   350.1 3102.54
   355.1 3103.53   411.8 3102.96   458.5 3104.79   507.8  3109.8   523.3 3113.99
#Mann= 4 ,-1,0
       0     .06       0      80      .1       0   148.1    .045       0
   172.8      .1       0
#XS Ineff= 2 , 0
          104.26  3103.9
Permanent Ineff=
       F       F
Bank Sta=148.1,172.8
XS Rating Curve= 0 ,0
Exp/Cntr=0.3,0.1

Type RM Length L Ch R = 1 ,28491   ,282.3,280.2,278.8
XS GIS Cut Line= 2
2325633.18838483602089.7633826042325308.91298433  602402.3981277
#Sta/Elev= 30
       0 3119.69    17.3 3118.62    20.1 3117.29      28 3110.98    39.9 3104.75
    62.5 3099.69    90.8 3097.24   102.9 3095.35   136.1 3094.55   155.9 3095.08
   160.5 3094.89   168.1 3093.34   175.7 3093.29     187 3092.71   195.1 3093.67
   223.8 3096.35   251.4 3095.64   262.6 3098.02   268.1 3098.23   279.2 3097.46
   318.1 3097.91   329.2 3096.61     357 3096.11   365.2 3094.92   379.2 3094.27
   395.9 3097.19     407 3097.34   416.2 3098.76   437.2 3105.48   450.4 3108.19
#Mann= 3 ,-1,0
       0      .1       0   175.7    .045       0   195.1      .1       0
Bank Sta=175.7,195.1
XS Rating Curve= 0 ,0
Exp/Cntr(USF)=0,0
Exp/Cntr=0.3,0.1

Type RM Length L Ch R = 1 ,28211   ,360.1,364.6,364.9
XS GIS Cut Line= 2
2325434.15591749601912.4634966542325165.55624483602240.087003044
#Sta/Elev= 30
       0 3112.22     6.1 3108.81    16.1 3108.93    24.7 3108.03    27.5  3106.8
      36 3099.96    44.5 3095.18    55.9 3091.09      63 3089.58    68.2 3089.83
    73.3 3091.38    78.5 3092.88      90 3094.32    99.2  3094.7   112.8 3091.48
   161.3 3090.96   175.3  3093.1   189.5 3093.16   255.5 3090.54   261.8 3090.89
   274.4  3094.8   306.1 3096.34   320.2 3093.26   348.7 3090.34   362.9 3091.65
   373.3  3096.8   382.8 3099.22   406.9  3103.9   414.7 3103.96   423.7 3105.57
#Mann= 4 ,-1,0
       0     .06       0    55.9    .045       0    73.3     .06       0
      90      .1       0
Bank Sta=55.9,73.3
XS Rating Curve= 0 ,0
Exp/Cntr=0.3,0.1

Type RM Length L Ch R = 1 ,27847   ,299.4,293.8,286.3
XS GIS Cut Line= 2
2325179.27383213 601705.651521142324843.35777623602161.300032609
#Sta/Elev= 30
       0 3105.61     4.7 3106.05    13.3 3105.35    25.4 3097.84    39.1 3093.91
    53.4 3088.62    72.6 3085.23    78.9 3085.74    93.8 3089.77   113.7 3089.58
   127.7 3086.41   182.1 3086.79   208.1 3085.88   218.1 3084.28   227.7    3084
   233.6 3084.31   239.3  3086.1   247.9 3087.44   262.8 3085.98   273.6  3086.6
   296.5 3089.81   322.4 3089.44   333.7 3086.78   342.3 3086.25   373.8 3090.26
   425.2 3089.98     504 3090.88   511.3 3091.51   537.7 3096.49   566.1 3097.72
#Mann= 4 ,-1,0
       0     .06       0     100      .1       0   208.1    .045       0
   239.3      .1       0
#XS Ineff= 2 , 0
                          313.62          3096.6
Permanent Ineff=
       F       F
Bank Sta=208.1,239.3
XS Rating Curve= 0 ,0
Exp/Cntr(USF)=0,0
Exp/Cntr=0.3,0.1

Type RM Length L Ch R = 1 ,27553   ,295.2,301.8,303.7
XS GIS Cut Line= 3
2324910.89476871601499.5688719022324749.86320478601908.833564295
2324734.27910258602183.039640981
#Sta/Elev= 30
       0 3109.64     6.4 3108.91    31.1 3098.51    44.7  3095.3    61.9 3088.16
    79.1 3087.19    86.6  3084.8    96.3 3083.47   104.9 3082.91   126.4 3084.45
   151.4 3082.06   216.7 3084.16   229.6 3081.23   240.9    3081     251 3080.55
   272.5 3081.08   321.1 3086.19   362.8 3086.61   410.1 3085.04   435.2 3087.17
   460.2 3085.06   476.2 3087.64   508.3 3089.03   532.7 3087.43   555.5 3087.27
   584.4 3088.39   652.5 3087.51   668.5    3089   688.1 3096.34   714.5 3100.29
#Mann= 3 ,-1,0
       0      .1       0   240.9    .045       0   272.5      .1       0
#XS Ineff= 2 , 0
                          326.96         3095.22
Permanent Ineff=
       F       F
Bank Sta=240.9,272.5
XS Rating Curve= 0 ,0
Exp/Cntr=0.3,0.1

Type RM Length L Ch R = 1 ,27251   ,345.5,329.2,313.6
XS GIS Cut Line= 2
2324774.91667624601378.1627249032324361.54037339601970.838379968
#Sta/Elev= 30
       0 3100.17    18.3 3098.66    24.2 3096.64    39.8 3093.96    47.2 3091.73
    55.8 3086.52    67.1 3085.41    87.5 3080.86   190.9 3079.22   226.8 3081.14
   257.3  3079.8     267 3081.11   282.8 3080.98   291.4 3079.85   319.4 3080.41
   333.4 3081.76   345.1 3080.53   379.2 3080.32   393.8 3079.14   417.3  3078.8
     428 3077.58   443.7 3078.89   460.9 3082.07   491.4 3083.53   515.7 3082.52
   662.1 3084.28   676.7 3086.08     690 3090.35     708 3094.33   722.6 3098.98
#Mann= 4 ,-1,0
       0     .06       0     140      .1       0   417.3    .045       0
   443.7      .1       0
#XS Ineff= 2 , 0
                          494.69          3087.8
Permanent Ineff=
       F       F
Bank Sta=417.3,443.7
XS Rating Curve= 0 ,0
Exp/Cntr(USF)=0,0
Exp/Cntr=0.3,0.1

Type RM Length L Ch R = 1 ,26922   ,392.7,425.8,432.9
XS GIS Cut Line= 3
2324480.51989525601187.5187897752324394.06232669 601325.85089947
 2324375.3298535601909.439487246
#Sta/Elev= 30
       0  3084.3    10.2 3083.64    21.8 3080.39    44.4 3081.74      68 3079.35
   106.3  3078.7   140.8 3079.67   190.5 3079.39   218.5  3080.4   222.5 3080.19
   242.5 3076.12   274.5 3077.07   284.5 3076.28   310.5 3075.75   315.5 3076.23
   394.6 3077.57   406.6 3076.68   426.6 3077.57   438.6 3076.24   458.2 3078.59
   501.7 3081.03   522.6  3080.3   534.6 3081.33   554.7 3081.12   574.7 3079.75
   590.7 3080.25   602.7 3081.63   634.7 3082.54   682.7 3082.54     747 3084.31
#Mann= 4 ,-1,0
       0     .06       0      50      .1       0   284.5    .045       0
   315.5      .1       0
#XS Ineff= 2 , 0
          220.33 3083.03
Permanent Ineff=
       F       F
Bank Sta=284.5,315.5
XS Rating Curve= 0 ,0
Exp/Cntr(USF)=0,0
Exp/Cntr=0.3,0.1

Type RM Length L Ch R = 1 ,26496   ,150.7,149.6,148
XS GIS Cut Line= 3
2324454.55292319601169.3217848232324335.63604087601337.044536549
2323992.76977102601655.807157444
#Sta/Elev= 30
       0 3084.14    13.1 3083.78    29.2 3080.91    83.2 3078.47   153.7 3078.24
     177 3079.33     196 3080.99   205.8 3082.76   211.7 3082.73   217.5 3082.34
   235.2 3078.24     241 3077.72   281.3  3078.8   295.9 3076.62   324.2 3075.75
     335 3076.35   357.8 3076.03   401.5  3072.5   443.1  3073.8   457.2 3072.27
   471.4 3073.81   479.9 3075.04   496.8 3075.82   521.6 3078.83   598.1  3077.7
   630.9 3078.73   638.4 3080.14   646.8  3083.7   663.6 3089.23   673.8 3091.65
#Mann= 4 ,-1,0
       0     .06       0      40      .1       0   443.1    .045       0
   471.4      .1       0
Bank Sta=443.1,471.4
XS Rating Curve= 0 ,0
Exp/Cntr=0.3,0.1

Type RM Length L Ch R = 1 ,26346   ,206.8,201.7,195.3
XS GIS Cut Line= 2
2324329.21915027601109.7069780712323872.43499638601583.782645672
#Sta/Elev= 30
       0 3085.05    20.2 3083.79    34.3 3076.44    41.9 3075.14   107.9 3074.66
   145.6 3076.29   162.9 3074.88   181.4 3075.93     204 3075.65     221 3074.09
   243.7 3075.47   257.8 3074.85   266.7 3072.28   297.4 3072.61   312.8 3073.73
   353.2 3072.29   365.3 3073.94   382.5 3072.48   399.2 3072.16   413.4 3072.44
   433.9 3072.38     453 3075.58     470 3076.09   520.3 3074.59   582.5 3074.75
   608.6 3081.67   619.9 3085.49   629.9 3086.82   639.7 3092.25   658.3 3099.97
#Mann= 4 ,-1,0
       0     .06       0     100      .1       0   382.5    .045       0
   413.4      .1       0
#XS Ineff= 2 , 0
          243.28 3077.78
Permanent Ineff=
       F       F
Bank Sta=382.5,413.4
XS Rating Curve= 0 ,0
Exp/Cntr(USF)=0,0
Exp/Cntr=0.3,0.1

Type RM Length L Ch R = 1 ,26145   ,304,324.5,342.4
XS GIS Cut Line= 3
2324167.68409448600959.471761365 2323944.7524296601195.383546594
2323790.71155563 601480.50103422
#Sta/Elev= 30
       0 3087.47    24.4 3086.32    29.2 3084.05    37.6 3077.71    46.1 3073.79
    95.9 3068.24   122.5 3070.03   150.8 3068.65   187.6 3070.37   255.5 3070.94
   292.3 3072.59   309.3    3072   332.2 3072.92   344.8 3072.37   372.1  3073.2
   379.5  3070.3   382.4  3069.2   390.3 3068.88   403.1 3070.08     413 3071.14
   450.3 3071.44   476.7 3070.49   490.3 3071.81   503.9 3070.99   535.8  3072.5
   556.6  3070.5   612.6 3071.23   618.6 3072.48   631.2 3079.94   648.6 3086.75
#Mann= 4 ,-1,0
       0     .06       0      60      .1       0   379.5    .045       0
   403.1      .1       0
Bank Sta=379.5,403.1
XS Rating Curve= 0 ,0
Exp/Cntr=0.3,0.1

Type RM Length L Ch R = 1 ,25820   ,315.8,319.3,316.2
XS GIS Cut Line= 3
2324060.51549071600865.9801859112323897.05993159600985.441885912
2323403.45104402601094.933364041
#Sta/Elev= 30
       0    3089    15.3 3088.63    25.2 3085.24    36.9 3082.97    69.8 3071.38
   100.3 3066.37   119.3 3065.96   139.1 3068.47   149.1 3067.46   178.8 3069.23
   215.7 3067.51   260.7 3069.38   286.1 3066.09   305.8 3064.26     317 3066.26
   334.5 3068.06   359.1 3068.08   371.3 3065.12   380.7 3067.15   404.1 3065.93
   424.6  3068.2   461.5 3065.41   473.8 3066.77   502.5 3065.76   518.8 3070.74
   633.6 3072.92   662.3 3077.97   682.7 3087.37     695  3091.2   708.1 3097.21
#Mann= 4 ,-1,0
       0     .06       0     120      .1       0   286.1    .045       0
     317      .1       0
Bank Sta=286.1,317
XS Rating Curve= 0 ,0
Exp/Cntr=0.3,0.1

Type RM Length L Ch R = 1 ,25501   ,372.9,382,387.5
XS GIS Cut Line= 4
2323989.11710164600692.565079122   2323843.85617600702.578152139
2323448.80692265600826.4651350072323265.27236935600824.404538405
#Sta/Elev= 30
       0 3089.37    49.1  3081.2   125.3  3072.5   145.6 3068.24     162 3066.62
   220.8 3065.81   258.5 3061.86   308.8 3063.58   346.5 3062.55   367.5 3060.78
     380 3061.25   383.6 3062.95   391.5 3065.81   405.2 3066.63   476.4 3066.88
   501.6 3071.31   518.4 3071.88   533.6 3069.23   556.1 3068.51   584.3 3071.35
   624.3 3070.55   632.3 3071.33   640.6 3073.69   676.3 3075.16   684.2 3076.41
   696.3 3080.64   708.7 3086.23   723.7 3094.79   736.3 3099.27   743.2 3103.29
#Mann= 4 ,-1,0
       0     .06       0      30      .1       0   346.5    .045       0
   383.6      .1       0
Bank Sta=346.5,383.6
XS Rating Curve= 0 ,0
Exp/Cntr=0.3,0.1

Type RM Length L Ch R = 1 ,25119   ,325.3,345.4,341
XS GIS Cut Line= 3
2323987.82496284600502.7348292722323912.39351583600460.828469823
2323271.84766713600481.101687455
#Sta/Elev= 30
       0 3080.68    53.8  3073.8    85.6 3068.47    94.5 3065.93   106.5 3063.85
   138.5 3063.68   222.6 3061.19   230.4 3059.81   239.1 3058.54   254.6 3058.63
   263.73059.704   294.6 3060.65   302.6 3061.63   330.6 3061.38   342.4 3062.14
   406.7 3060.24   445.7 3063.52   474.7 3062.53   498.7 3060.35   514.7 3061.63
   534.7 3061.01   554.7 3059.05   570.8 3059.78   602.8 3063.66   646.8 3063.78
   658.8 3064.88   678.8 3069.75   698.8 3076.28   706.8 3077.54   727.2 3086.63
#Mann= 4 ,-1,0
       0     .06       0      30     .12       0   230.4    .045       0
   263.7      .1       0
#XS Ineff= 2 , 0
          136.04 3072.67  600.58         3070.72
Permanent Ineff=
       F       F
Bank Sta=230.4,263.7
XS Rating Curve= 0 ,0
Exp/Cntr(USF)=0,0
Exp/Cntr=0.3,0.1

Type RM Length L Ch R = 1 ,24773   ,313.7,326.7,328
XS GIS Cut Line= 3
2324004.36613837600212.1490308712323765.82924748600282.417509843
2323232.73460109 600336.94844023
#Sta/Elev= 30
       0 3072.44     8.5 3072.85      21 3071.91      30 3067.28    37.7  3065.7
   225.4 3061.16   246.2 3062.39   254.4 3061.72   274.5 3057.74   296.7 3059.85
   350.9  3060.8   399.1 3059.43   420.5 3060.36   435.3 3058.12     446 3060.14
   475.5 3060.16   516.2 3057.17   539.8 3056.31   559.9 3056.97     568 3056.69
     580 3057.91   588.3 3056.81   604.2 3060.63   632.3  3062.5   672.2 3062.82
   688.6 3064.06   716.8  3072.4   744.9 3078.62   770.7 3087.22   784.5  3093.6
#Mann= 5 ,-1,0
       0     .06       0     150     .12       0  348.67      .1       0
   516.2    .045       0   559.9      .1       0
#XS Ineff= 2 , 0
           245.8 3071.31
Permanent Ineff=
       F       F
Bank Sta=516.2,559.9
XS Rating Curve= 0 ,0
Exp/Cntr=0.3,0.1

Type RM Length L Ch R = 1 ,24447   ,417.8,415.5,406.3
XS GIS Cut Line= 3
2323979.27441218600023.4865907392323802.72699416600062.688409261
2323206.35045688599949.990059249
#Sta/Elev= 30
       0 3083.09    11.4 3080.59    23.7  3071.9    27.5 3070.39    48.2 3069.92
    52.3 3068.79    60.5 3063.65    64.6 3062.11     163 3061.03   276.8 3058.44
   305.6  3056.7   338.1  3056.5   350.3 3057.41   362.4 3054.79   378.8 3053.11
   406.9  3054.6   423.6 3056.71   439.9 3056.25   460.3 3058.49   492.8 3057.38
   549.8 3057.41   606.8 3059.07   651.6  3062.5     676 3062.41   684.2 3062.97
   688.2 3064.32   696.4 3070.36   700.4 3071.86   752.7 3075.14   787.8  3079.9
#Mann= 6 ,-1,0
       0      .1       0      20     .06       0     120     .12       0
  220.85      .1       0   362.4    .045       0   406.9      .1       0
#XS Ineff= 2 , 0
           274.4 3064.02
Permanent Ineff=
       F       F
Bank Sta=362.4,406.9
XS Rating Curve= 0 ,0
Exp/Cntr=0.3,0.1

Type RM Length L Ch R = 1 ,24031   ,369.6,372.9,379.6
XS GIS Cut Line= 2
2323926.55591665599647.8340202872323219.99996011599686.565051085
#Sta/Elev= 30
       0 3062.75     6.4 3060.02    10.4 3058.98    22.3 3058.13   110.5 3056.48
   150.6 3057.46   234.7 3055.16   238.7 3054.58   246.6 3050.95   254.2 3049.73
   266.8 3049.28   274.8 3050.58   290.8  3050.9   314.9 3049.88   362.9 3049.67
   378.9 3051.17   390.9 3050.63     395 3050.99     415 3054.64   503.1 3054.65
   547.2 3055.88   555.2 3057.18   581.7 3067.39   602.9 3071.23   607.3 3071.52
   615.3 3070.88   627.3 3071.57   643.3 3073.19   691.4 3076.14   707.6 3077.97
#Mann= 5 ,-1,0
       0     .06       0      60     .12       0     160      .1       0
   246.6    .045       0   274.8      .1       0
#XS Ineff= 2 , 0
                          416.62         3060.63
Permanent Ineff=
       F       F
Bank Sta=246.6,274.8
XS Rating Curve= 0 ,0
Exp/Cntr=0.3,0.1

Type RM Length L Ch R = 1 ,23658   ,351.1,349.9,353.4
XS GIS Cut Line= 3
2323917.90129091 599305.723442122323742.11907958  599351.7905044
2323265.68867232599362.701124414
#Sta/Elev= 30
       0 3063.03    14.2 3060.83    22.5 3057.02    33.7 3054.21      39 3053.71
   135.3 3051.49   179.6 3052.62   195.7 3049.67   216.3    3050   235.7 3048.99
   251.7 3050.66   282.8 3051.44   295.7 3048.24   303.7 3047.81   319.7 3048.92
   399.7 3050.54   432.1 3047.39   451.7 3046.16   467.7  3046.3   475.63047.982
   483.7 3052.78   487.7 3053.21   535.8 3051.85   555.8  3048.4   583.8 3049.94
   591.8 3052.91   603.5 3062.54   624.5 3077.02   628.6 3078.43   658.3 3083.37
#Mann= 4 ,-1,0
       0     .06       0      60      .1       0   432.1    .045       0
   475.6      .1       0
#XS Ineff= 2 , 0
          180.58 3062.28
Permanent Ineff=
       F       F
Bank Sta=432.1,475.6
XS Rating Curve= 0 ,0
Exp/Cntr(USF)=0,0
Exp/Cntr=0.3,0.1

Type RM Length L Ch R = 1 ,23308   ,348.5,346.6,340.5
XS GIS Cut Line= 2
2323868.96772591599037.0744826892323273.11495954599062.618987486
#Sta/Elev= 30
       0 3069.05    20.8 3067.14    32.8    3061    52.8 3062.21      76 3050.86
    88.9  3048.9   104.9 3048.26   160.9 3050.13     173 3048.49     201 3048.42
     209 3046.81     225 3047.93   231.2 3046.28     237 3044.47     261 3044.44
   269.6 3045.52   301.1 3044.89   313.1 3047.32   329.1 3048.53   365.1 3048.79
   397.2 3047.34   429.2 3048.98   457.2 3048.21   485.2 3045.48   499.9 3047.39
   513.3 3045.37   525.3 3045.94   530.7 3046.94   573.3 3066.86   596.4 3070.56
#Mann= 5 ,-1,0
       0      .1       0      10     .06       0     110      .1       0
   231.2    .045       0   269.6      .1       0
#XS Ineff= 2 , 0
          158.84 3058.43
Permanent Ineff=
       F       F
Bank Sta=231.2,269.6
XS Rating Curve= 0 ,0
Exp/Cntr=0.3,0.1

Type RM Length L Ch R = 1 ,22962   ,232.4,239.4,241.7
XS GIS Cut Line= 3
2323887.17321819598648.1421138922323793.36878181598670.598181477
2323189.83726158598796.454295369
#Sta/Elev= 30
       0 3062.15    27.8 3061.41    48.3 3056.31    56.6 3056.25    77.1 3052.31
   126.7 3047.35   171.2 3046.03     208 3047.34   212.1 3047.01   220.3 3043.44
   232.5 3043.62   240.7 3041.93   265.9 3042.64   277.5 3040.66   289.7 3040.93
   297.9 3042.84   306.1 3044.38   339.7 3043.53   383.6 3046.47   404.1 3043.09
   424.6 3042.53   525.7  3045.1   559.3 3043.74   596.2    3045   610.2 3043.12
     637 3043.89   645.2 3047.28   657.5 3058.22   673.8 3069.58     713 3085.46
#Mann= 4 ,-1,0
       0     .06       0      30      .1       0   265.9    .045       0
   297.9      .1       0
#XS Ineff= 2 , 0
           208.7 3057.48
Permanent Ineff=
       F       F
Bank Sta=265.9,297.9
XS Rating Curve= 0 ,0
Exp/Cntr=0.3,0.1

Type RM Length L Ch R = 1 ,22722   ,459.9,462.5,454.1
XS GIS Cut Line= 3
2323826.54794894598463.8899101432323656.92697022598490.497122492
2323156.37878791598502.137777894
#Sta/Elev= 30
       0 3057.91      55 3049.37   111.7    3047   180.4 3045.44   204.5 3045.96
   232.5 3045.31   251.6 3041.35   264.5 3041.84   280.3 3040.44   288.5 3039.09
   304.5 3039.12   308.5 3039.51   312.5 3041.54   320.5 3042.93   368.5 3043.28
   380.5 3039.75   412.5 3038.93   440.5  3040.2   452.5 3042.24   468.5 3041.39
   487.9 3042.24   520.5 3041.59   540.5 3042.77   588.6 3041.49   608.6 3045.03
   624.6 3051.67   636.4 3058.78   644.6 3062.71   656.6 3071.48   672.4 3079.48
#Mann= 4 ,-1,0
       0     .06       0      60      .1       0   280.3    .045       0
   312.5      .1       0
Bank Sta=280.3,312.5
XS Rating Curve= 0 ,0
Exp/Cntr(USF)=0,0
Exp/Cntr=0.3,0.1

Type RM Length L Ch R = 1 ,22260   ,285.2,284.8,287.9
XS GIS Cut Line= 3
 2323671.7484921598158.584584896 2323207.1455996598260.666492282
2323074.22894507598328.145598348
#Sta/Elev= 30
       0 3049.54    24.1 3046.17    42.1 3047.66    55.5 3046.46    65.1 3047.12
    77.4  3046.5    85.8 3045.32    97.9 3041.52     106 3040.56   175.7 3041.16
   193.2 3039.05   245.3 3037.95   278.1 3039.57   324.2 3038.39   335.4 3036.47
   355.9 3036.49   361.1 3038.29   364.1 3039.83   372.2 3040.51   510.4 3040.24
   523.9 3038.72   546.7 3038.99   550.8 3039.85   561.6 3045.14     574 3054.02
   586.7 3060.74   597.3 3067.59   604.6 3070.83   618.1 3081.51   624.8 3083.97
#Mann= 4 ,-1,0
       0     .06       0     110      .1       0   324.2    .045       0
   361.1      .1       0
Bank Sta=324.2,361.1
XS Rating Curve= 0 ,0
Exp/Cntr=0.3,0.1

Type RM Length L Ch R = 1 ,21975   ,328.4,312.9,307.8
XS GIS Cut Line= 3
2323470.72576233597921.1427188982323269.99009484597958.533359746
2322973.45524293598099.849536752
#Sta/Elev= 30
       0 3048.79    10.7 3049.73    51.4 3048.81    81.1 3047.15   104.3  3047.6
   108.4 3046.56   120.6 3036.38   124.7 3034.86   128.7 3034.43   140.9 3034.34
   153.7 3035.55   173.7 3037.67   210.6 3039.44   237.2  3038.5     348 3038.46
   352.4 3038.02   356.9 3035.67   361.3 3034.62     379 3036.55   396.7 3035.71
   405.6 3036.31   432.2 3034.45   436.6  3035.4   441.6 3037.71   450.6 3039.17
   461.4 3045.07   474.6  3049.4   504.6 3062.41   520.8 3067.78   532.7 3072.95
#Mann= 4 ,-1,0
       0     .06       0     100      .1       0   120.6    .045       0
   153.7      .1       0
Bank Sta=120.6,153.7
XS Rating Curve= 0 ,0
Exp/Cntr=0.3,0.1

Type RM Length L Ch R = 1 ,21662   ,402.7,393.8,389.9
XS GIS Cut Line= 2
2323253.40044423597638.3482564442322865.16273261597903.484800027
#Sta/Elev= 30
       0 3044.31    25.9 3045.65    45.1 3042.69    61.8 3041.52    89.3 3041.11
   112.3 3042.32   117.7 3040.99   123.8 3037.27   127.4 3036.05   137.1 3034.78
     154 3034.99   156.5 3034.36   161.2 3032.14   166.2  3031.6   180.7 3031.47
   190.4 3031.56   195.8 3032.26   203.6 3034.12   207.3 3034.52   248.5 3034.69
   267.4 3037.11   279.2 3037.68     310    3037   333.9 3037.54   345.4 3036.53
   364.8 3036.11   402.2 3039.85   409.3 3041.47   422.9 3046.19   470.1 3065.76
#Mann= 4 ,-1,0
       0     .06       0     100      .1       0   161.2    .045       0
   195.8      .1       0
Bank Sta=161.2,195.8
XS Rating Curve= 0 ,0
Exp/Cntr(USF)=0,0
Exp/Cntr=0.3,0.1

Type RM Length L Ch R = 1 ,21268   ,237.4,238.9,236.5
XS GIS Cut Line= 3
2323149.90320637597559.5364321822322892.10771335597475.047794802
2322675.43683485597706.159957527
#Sta/Elev= 30
       0    3040   132.3 3035.46   278.4 3034.15   290.7 3033.57   306.7 3034.27
   318.1 3033.18     352 3032.98   372.9 3031.41   382.3 3032.02   388.8 3031.51
   394.8 3032.58   405.8 3033.03   434.9 3030.53   445.4 3031.67   460.6 3031.63
     468 3030.72   471.6 3029.61   477.1 3029.31   493.5 3029.31     499 3029.97
   500.4 3030.76     510 3038.58   516.1 3044.54   520.9 3050.93   526.4 3055.42
   544.4 3065.34   559.3  3072.8   567.1 3075.63   578.4 3082.06   588.1 3085.68
#Mann= 4 ,-1,0
       0     .06       0  291.29      .1       0     468    .045       0
   500.4      .1       0
Bank Sta=468,500.4
XS Rating Curve= 0 ,0
Exp/Cntr=0.3,0.1

Type RM Length L Ch R = 1 ,21029   ,169.7,207,240.7
XS GIS Cut Line= 4
2323156.96375855597505.5012904922322896.72175095597454.206846129
2322693.75754409597395.8027341782322574.23287937  597527.1237447
#Sta/Elev= 30
       0 3043.54    25.3 3041.13    78.3 3038.76    89.5 3036.08    94.6  3035.4
   123.1 3034.02   143.5 3034.43     172 3032.34   180.2 3032.22   192.4 3032.97
   208.7 3032.03   229.1 3032.88   249.6 3032.43   261.7 3034.04   324.1 3034.13
     370 3033.78     449 3031.28   483.7 3032.53   502.6 3030.29   505.4 3029.71
   509.7 3027.72   516.2  3026.9   526.3 3026.85   540.8  3027.6   556.1 3029.73
   597.5 3028.92   609.5 3032.54   614.5 3034.66   634.3 3049.68     654 3067.75
#Mann= 4 ,-1,0
       0     .06       0   509.7    .045       0   540.8     .06       0
  556.45      .1       0
#XS Ineff= 2 , 0
          274.59  3046.7
Permanent Ineff=
       F       F
Bank Sta=509.7,540.8
XS Rating Curve= 0 ,0
Exp/Cntr(USF)=0,0
Exp/Cntr=0.5,0.3

Type RM Length L Ch R = 1 ,20822   ,50.1,55.2,69.8
XS GIS Cut Line= 4
2323138.51337228597481.2296027352322704.79324651597386.520766561
2322469.66929101597175.1008066092322429.05633445597184.259298011
#Sta/Elev= 30
       0 3041.24    49.1 3039.51    92.5  3034.8   108.8 3035.08   149.8 3032.62
     170 3032.42   190.7 3031.75   260.3 3032.01   280.8 3030.42     289 3032.61
   297.7 3033.48     375 3033.13   440.5 3030.92   450.2 3031.37   499.1 3028.81
   511.8 3029.61   573.9 3027.83   584.6 3029.56   609.6 3026.07   613.5 3024.85
   620.9 3024.46   632.3 3024.73   635.1 3025.99   638.4 3028.12   643.4 3029.33
   659.9  3027.8   670.7 3027.95   760.1 3031.12   786.5 3044.41   801.8  3049.9
#Mann= 5 ,-1,0
       0     .06       0     130      .1       0     170     .06       0
   609.6    .045       0   635.1     .06       0
#XS Ineff= 2 ,-1
     290     583  3026.3     643     800  3026.4
Permanent Ineff=
       F       F
Bank Sta=609.6,635.1
XS Rating Curve= 0 ,0
Exp/Cntr=0.5,0.3

Type RM Length L Ch R = 1 ,20767   ,150.7,115,81.4
XS GIS Cut Line= 5
2323162.96033052 597440.770044792322723.03813355597338.760106814
2322539.98217555597170.2516421592322469.66929101 597110.84937764
2322406.76007426 597129.41743474
#Sta/Elev= 30
       0 3040.79    43.9 3039.91    88.6 3036.67   150.7  3034.4   183.5 3035.42
   204.1 3034.22   220.5 3032.21   294.4 3032.74   335.5 3031.78   376.5 3029.28
   440.9 3030.99   526.2 3029.68   569.7 3027.98   583.9 3026.13   591.4 3026.18
   596.8 3024.42   601.6 3023.72   630.3 3023.43   662.1 3023.59   666.5 3024.26
   672.7  3026.4   683.8 3028.39   720.7 3028.85   731.6 3031.73   736.8 3032.21
   792.4 3031.25   827.7 3032.61   840.6 3032.11   844.1 3032.68     858  3039.2
#Mann= 9 ,-1,0
       0      .1       0     190     .06       0     380      .1       0
     390     .06       0  581.59      .1       0   596.8    .045       0
   666.5     .06       0   720.4      .1       0   770.4     .06       0
#XS Ineff= 3 ,-1
     321     435    3033     435     580  3026.3     675     800  3026.4
Permanent Ineff=
       F       F       F
Bank Sta=596.8,666.5
XS Rating Curve= 0 ,0
Exp/Cntr(USF)=0,0
Exp/Cntr=0.5,0.3

Type RM Length L Ch R = 1 ,20652   ,68,66.9,65.6
XS GIS Cut Line= 3
2323049.57701334597014.4102678862322622.28304659597100.398095388
2322415.24144627597104.065134376
#Sta/Elev= 30
       0 3036.13     9.6 3034.21    25.9  3034.1    38.2 3032.85   122.4 3031.81
   136.1 3030.65   189.1 3029.07   225.8 3029.26   242.2 3027.85   270.7 3030.11
   299.3 3026.66   319.7 3025.53   356.4    3028   364.6 3027.09   380.9  3027.2
   393.1 3025.67   413.5 3026.66   433.9 3029.37   458.4 3027.48     466  3026.2
   470.1 3024.65   485.9 3023.31     502 3023.46   510.5 3024.61     518 3026.99
     522 3027.23     530 3025.39     546 3028.57     558  3029.9   642.9 3033.46
#Mann= 6 ,-1,0
       0      .1       0      70     .12       0     240      .1       0
   470.1    .045       0   510.5      .1       0  575.86     .06       0
Bank Sta=470.1,510.5
XS Rating Curve= 0 ,0
Exp/Cntr(USF)=0,0
Exp/Cntr=0.3,0.1
